--- War Creek.prj (project) ---

Proj Title=War Creek
Current Plan=p01
Default Exp/Contr=0,0
English Units
Geom File=g01
Flow File=f01
Plan File=p01
BEGIN DESCRIPTION:
END DESCRIPTION:
DSS Export Rating Curves= 0
DSS Export Rating Curve Sorted= 0
DSS Export Volume Flow Curves= 0
DXF OffsetX= 0
DXF OffsetY= 0
DXF ScaleX= 0
DXF ScaleY= 0

--- War Creek.p01 (plan) ---

Plan Title=Floodplain
Program Version=4.00
Geom File=g01
Flow File=f01
K Sum by GR=0
Std Step Tol=0.01
Critical Tol=0.01
Num of Std Step Trials=20
Max Error Tol=0.3
Flow Tol Ratio=0.001
Split Flow NTrial=30
Split Flow Tol=0.02
Split Flow Ratio=0.02
Log Output Level=0
Friction Slope Method=1
Unsteady Friction Slope Method=2
Unsteady Bridges Friction Slope Method=1
Global Log Level=0
CheckData=False
Run HTab=0
Run UNet=0
Run PostProcess=0
UNET Theta=0
UNET Theta Warmup=0
UNET ZTol=0
UNET ZSATol=0
UNET MxIter=0
UNET MaxInSteps=0
UNET DtIC=0
UNET DtMin=0
UNET MaxCRTS=0
UNET WFStab=0
UNET SFStab=0
UNET WFX=0
UNET SFX=0
UNET DSS MLevel=0
UNET DZMax Abort=0
UNET Convert EG Bridges=0
UNET Use Existing IB Tables=0
UNET Froude Limit=0
UNET Froude Power=0
Write IC File=0
Echo Input=False
Echo Output=False
Write Detailed=0

--- War Creek.f01 (steady flow) ---

Flow Title=NFF Regression Equation
Program Version=4.00
Number of Profiles=1
Profile Names=P100yr
River Rch & RM=War Creek,Main      ,16206.7
576.1014
River Rch & RM=War Creek,Main      ,15208.6
1646.326
River Rch & RM=War Creek,Main      ,12246
1741.968
River Rch & RM=War Creek,Main      ,11476.7
1769.675
Boundary for River Rch & Prof#=War Creek,Main      ,1
Up Type=0
Dn Type=3
Dn Slope=0.012392

--- War Creek.g01 (geometry) ---

Geom Title=USGS 10m DEM
Program Version=4.00

River Reach=War Creek       ,Main
Reach XY= 30
     1764128.886       94597.019      1764469.79       95308.927
     1764891.196       95089.669     1765279.082         95085.2
     1766377.496       95898.509     1766564.289       95865.441
     1766593.783       96257.795      1766738.57       96424.032
     1766773.426        96664.45     1766557.217       97308.505
     1766775.213        97523.34     1766898.631       98129.206
     1767386.524       98306.043     1767859.208       99272.578
     1768544.093       99443.726     1768114.068      100834.241
     1768285.273      101232.379     1767936.023      101368.374
     1767858.721      101530.959     1767552.504      101739.924
     1767060.762      102815.673     1766429.377      103126.877
     1766563.035      103349.308     1766497.594      103442.082
     1766672.255      103541.816     1766632.856      103761.255
     1766868.254      104564.699     1767038.818      104848.973
     1766878.727      105625.486     1766655.236      105792.322

Type RM Length L Ch R = 1 ,16206.7 ,248.1,259.2,270.3
XS GIS Cut Line= 4
     1763732.137       94836.377     1764088.911       94690.228
     1764312.432        94402.23     1764355.417       94217.395
#Sta/Elev= 30
     2.9  1751.4      16 1742.73    26.2 1742.73    37.9 1732.65    59.7 1729.36
    70.6 1718.18    81.6 1717.89   103.4 1707.26   223.7 1690.91   234.6 1688.21
   245.5 1678.04   278.3  1668.4   388.7 1656.17   480.2 1650.17   487.7 1649.81
   495.2 1649.82   570.2 1664.16   586.7 1660.91   609.2 1667.64   636.2 1663.86
   652.7 1671.76   673.2 1664.87   698.8  1672.4   711.6 1664.06   718.7 1664.06
   737.2 1674.02   798.9 1670.11   843.5 1678.93   895.4 1675.81   939.9 1684.73
#Mann= 3 , 0 , 0
     2.9     .08       0   480.2    .045       0   495.2     .08       0
Bank Sta=480.2,495.2
XS Rating Curve= 0 ,0
Exp/Cntr=0.3,0.1

Type RM Length L Ch R = 1 ,15947.5 ,407.2,404.5,401.9
XS GIS Cut Line= 4
     1763925.409       95072.561     1764101.806       94900.854
     1764389.805       94763.303     1764644.043       94637.439
#Sta/Elev= 30
     3.8 1776.87    33.3 1769.03    47.3 1750.88    75.6 1747.22    90.8 1729.88
   103.8    1729   146.2 1708.25   160.3 1694.91   174.4 1692.63   192.3 1679.62
   221.4 1675.22   235.9 1665.58   357.3  1649.8   386.9 1649.79   458.2 1649.85
   491.8 1653.81   525.5 1663.53   536.7 1671.67   615.5 1693.67   626.7 1704.96
   638.1 1705.36   660.6    1719     672 1719.12   683.2 1733.61   705.8 1740.04
   717.1 1751.82   762.2  1764.2   773.5 1775.71   818.7 1787.49     849 1801.39
#Mann= 3 , 0 , 0
     3.8     .08       0   357.3    .045       0   458.2     .08       0
Bank Sta=357.3,458.2
XS Rating Curve= 0 ,0
Exp/Cntr=0.3,0.1

Type RM Length L Ch R = 1 ,15543   ,371.8,334.4,305.3
XS GIS Cut Line= 4
     1760365.587       95195.526     1764100.256       95398.647
     1764580.107         95094.1     1764759.474       94526.886
#Sta/Elev= 30
     2.9 2204.45   124.5 2235.47   266.3 2215.26   458.8 2114.42     631 2000.23
   742.4 1957.29   782.9 1966.74   985.5 2092.79    1026 2085.96  1117.2 2026.72
  1208.4 2004.71  1583.2 2162.46  1755.4 2091.09  2008.7 1942.43  2069.4 1933.06
  2332.8 2036.93  2494.9 2077.17  2687.4 2102.61  2808.9 2094.44  2889.3 2073.92
  2981.1 2003.32  3214.1 1956.95  3548.4 1763.19    3741 1693.73  3932.7 1649.81
  3969.2 1649.78  4259.3  1649.8  4461.2 1694.73  4832.9    1870  4903.4 1888.64
#Mann= 3 , 0 , 0
     2.9     .08       0  3932.7    .045       0  4259.3     .08       0
Bank Sta=3932.7,4259.3
XS Rating Curve= 0 ,0
Exp/Cntr=0.3,0.1

Type RM Length L Ch R = 1 ,15208.6 ,289.5,293.2,296.9
XS GIS Cut Line= 4
     1762804.405       99417.567     1764797.819       95532.477
     1764587.596       95089.419     1764764.017       94616.451
#Sta/Elev= 30
       4 2313.46   159.1 2278.72     425 2295.01   623.2 2217.11  1023.2 2132.01
  1600.4 2193.05  1714.7  2166.3  1771.5 2121.76  1907.9 2082.85  2153.3 1919.39
  2226.3 1881.28  2305.8 1866.03  2662.9 1920.68  2931.1 2058.09  3010.7 2022.11
  3022.1 2001.34  3101.7 1948.27  3215.3 1898.06  3431.4  1889.1    3636 1783.66
  3704.2 1781.09    3852 1831.54  3999.8 1839.55  4113.5 1794.66    4284 1696.85
  4552.2  1649.8  4668.3 1649.77  4822.7  1649.8  5039.8 1706.18  5361.9  1852.4
#Mann= 3 , 0 , 0
       4     .08       0  4552.2    .045       0  4822.7     .08       0
Bank Sta=4552.2,4822.7
XS Rating Curve= 0 ,0
Exp/Cntr=0.3,0.1

Type RM Length L Ch R = 1 ,14915.4 ,202.6,209.1,215.7
XS GIS Cut Line= 4
     1764943.772       95628.372     1764986.592       95361.981
     1764857.802       94929.869     1764873.921       94462.409
#Sta/Elev= 30
     2.2 1754.08     107 1768.75   176.3 1766.77   279.1 1727.03   300.2 1707.22
   321.3 1700.44   331.8 1686.01   352.9 1686.01   363.5 1669.68   405.7  1649.8
   553.5 1649.76   663.6 1649.82   752.7 1692.59   803.3 1705.16   853.9 1742.76
   874.1 1742.75   884.2 1758.99   904.5  1760.3   955.1 1797.28   975.3 1797.21
   985.4 1814.53  1005.7 1815.94  1056.3 1852.04  1076.2 1851.94  1086.7 1869.94
  1106.9 1871.63  1147.4 1899.44  1157.5 1913.82  1177.7  1913.9  1188.4 1930.62
#Mann= 3 , 0 , 0
     2.2     .08       0   405.7    .045       0   663.6     .08       0
Bank Sta=405.7,663.6
XS Rating Curve= 0 ,0
Exp/Cntr=0.3,0.1

Type RM Length L Ch R = 1 ,14706.3 ,28.8,28.9,29
XS GIS Cut Line= 3
     1765072.726       95612.253     1765113.294       95214.162
     1765088.845       94467.782
#Sta/Elev= 30
     6.3 1828.15   128.3 1814.78   138.5 1797.72   199.5  1773.8   209.6 1759.85
     230 1759.94   280.8 1723.76   301.2 1720.97   311.3 1705.61   331.7 1705.56
   412.9 1656.09   514.5 1649.81   554.5 1649.75   673.3 1649.87     767 1656.63
   807.4 1674.15   817.5 1689.64   837.8 1689.61   847.9 1704.54   868.2 1709.52
   888.5  1729.2   908.8 1731.73   918.9 1748.24   939.2 1747.64   949.4 1761.68
  1010.3 1786.67  1020.4 1802.12  1040.7 1802.11  1050.8 1814.85  1147.5 1859.13
#Mann= 3 , 0 , 0
     6.3     .08       0   514.5    .045       0   673.3     .08       0
Bank Sta=514.5,673.3
XS Rating Curve= 0 ,0
Exp/Cntr=0.3,0.1

Type RM Length L Ch R = 1 ,14677.4 ,12.7,12.7,12.7
XS GIS Cut Line= 3
     1765102.736       95604.827      1765141.45       95256.396
     1765134.411       94499.704
#Sta/Elev= 30
     7.8 1841.31      81 1835.39   100.6 1818.66     121 1819.68   131.1 1803.47
   192.2 1777.98   202.4 1761.78   222.7 1761.78   273.6  1722.5     294 1719.88
   304.1 1703.92   324.5 1703.61   405.6 1659.14   669.8 1650.29   677.3 1649.61
   684.8 1649.62   759.6 1654.62   800.1 1672.91   810.2 1691.31   830.4 1691.22
   840.5  1707.5     881 1735.13   901.3 1737.61   911.4 1755.92   931.6 1755.64
   982.2 1793.44  1002.4 1795.55  1012.5 1811.47  1032.8 1811.24  1107.3 1851.16
#Mann= 3 , 0 , 0
       0     .08       0   669.8    .045       0   684.8     .08       0
Bank Sta=669.8,684.8
XS Rating Curve= 0 ,0
Exp/Cntr=0.3,0.1

Type RM Length L Ch R = 1 ,14664.7 ,8.4,8.8,9.2
XS GIS Cut Line= 3
     1765118.911       95604.827     1765154.106        95231.76
     1765150.587       94489.145
#Sta/Elev= 30
     2.3 1847.98    48.7 1852.05    90.3 1838.01   100.4 1822.45   120.7 1822.45
   171.5 1781.03   191.9 1778.95     202 1762.61   222.3 1762.96   273.2 1721.38
   293.5  1718.9   303.6  1702.6     324 1702.39   405.1 1659.39   671.9 1650.18
   679.4 1649.46   686.9 1649.47   759.1 1654.46   799.6 1672.77   809.7 1692.09
   829.9 1692.07   880.5  1737.1   900.7 1739.64   910.9 1758.58   931.1 1758.58
   981.7 1797.49  1001.9 1799.69    1012 1815.91  1032.2 1815.91  1117.4 1864.47
#Mann= 3 , 0 , 0
     2.3     .08       0   671.9    .045       0   686.9     .08       0
Bank Sta=671.9,686.9
XS Rating Curve= 0 ,0
Exp/Cntr=0.3,0.1

Type RM Length L Ch R = 1 ,14655.9 ,24.2,23.8,23.4
XS GIS Cut Line= 3
     1765143.477       95437.364     1765161.561        95169.74
     1765164.606       94982.284
#Sta/Elev= 30
     2.5 1783.67    23.6 1780.69    33.8 1763.96      54 1764.25    64.2 1748.64
    84.4 1742.63   104.7 1720.84     125 1718.48   135.1 1702.06   155.4 1702.02
   165.5 1689.33   226.4 1669.21   236.5 1659.39   551.2 1649.12   558.7  1649.1
   561.9 1650.11   631.1 1674.13   641.2 1693.79   661.4 1693.86   671.6 1710.33
   691.8 1717.08     712 1739.59   732.3 1742.11   742.4 1761.52   762.6 1761.62
   772.7 1776.23   792.9 1782.25   813.2 1800.96   833.4  1803.1   842.5 1817.78
#Mann= 3 , 0 , 0
     2.5     .08       0   551.2    .045       0   561.9     .08       0
Bank Sta=551.2,561.9
XS Rating Curve= 0 ,0
Exp/Cntr=0.3,0.1

Type RM Length L Ch R = 1 ,14632.1 ,18.7,19.3,20
XS GIS Cut Line= 3
      1765153.45        95393.88     1765186.691       95129.024
     1765190.771       94563.254
#Sta/Elev= 30
    10.5 1765.32    20.7 1749.12    41.1 1742.73    61.5 1720.62    81.9 1718.31
    92.1 1701.13   112.4 1699.87   122.6 1686.96   163.4  1666.5   285.6 1646.58
   301.7 1635.61   309.2 1635.57   316.7 1636.42   336.2 1652.05   366.5 1655.97
   493.5 1647.03   548.6 1657.66   568.8  1676.6   589.1 1678.85   599.2  1699.1
   619.4 1699.33   629.5 1715.74   649.8 1723.05     670 1746.17   690.2 1748.44
   700.3 1768.64   720.6 1768.92   737.3 1787.86   791.4  1810.5   832.7 1838.46
#Mann= 3 , 0 , 0
       0     .08       0   301.7    .045       0   316.7     .08       0
Bank Sta=301.7,316.7
XS Rating Curve= 0 ,0
Exp/Cntr=0.3,0.1

Type RM Length L Ch R = 1 ,14612.8 ,66.7,78.3,89.8
XS GIS Cut Line= 4
      1765130.69       95604.607     1765204.041       95154.587
     1765209.531       94965.863     1765214.272       94561.378
#Sta/Elev= 30
     8.8 1851.45    49.8  1853.2    90.8  1839.1   101.1 1824.55   121.6 1825.24
   172.8 1784.95   193.3 1782.72   203.6 1765.24   224.1 1764.57   275.3 1717.04
   295.8 1714.84   306.1 1696.91   326.6 1696.76   408.5 1652.45     513 1627.11
   522.9 1627.01     528 1627.02   581.2 1649.65   702.6 1645.46   763.3 1660.46
   783.5 1680.83   803.7 1682.62   813.9 1702.84   834.1 1703.29   884.7 1750.24
   904.9 1752.03     915 1772.37   934.5 1772.85   955.5 1793.81  1049.3 1842.44
#Mann= 3 , 0 , 0
     8.8     .08       0     513    .045       0     528     .08       0
Bank Sta=513,528
XS Rating Curve= 0 ,0
Exp/Cntr=0.3,0.1

Type RM Length L Ch R = 1 ,14534.5 ,352.9,346.4,339.9
XS GIS Cut Line= 4
     1765196.307       95773.446     1765195.698       95248.609
     1765421.978       94833.153     1765405.858       94526.886
#Sta/Elev= 30
     5.6 1873.21   116.9 1875.86     218    1855   238.3 1838.56   258.5 1836.88
   268.6    1820   288.8 1819.73   339.4 1781.15   359.6 1779.12   369.8 1760.04
     390 1759.74   440.6 1714.26   460.8 1712.35   470.9 1694.14   491.1 1693.87
   544.1  1658.6   613.2 1632.55   702.9 1623.85   710.4  1623.7   717.9 1624.46
   739.9 1636.26   797.5 1636.46     855 1660.85   900.7 1655.48    1004 1723.69
  1024.2 1723.69  1034.3 1737.57  1054.6 1740.21  1105.2 1772.46  1304.6 1826.36
#Mann= 3 , 0 , 0
       0     .08       0   702.9    .045       0   717.9     .08       0
Bank Sta=702.9,717.9
XS Rating Curve= 0 ,0
Exp/Cntr=0.3,0.1

Type RM Length L Ch R = 1 ,14188.1 ,110.7,109.3,107.9
XS GIS Cut Line= 4
     1765385.092       95676.903     1765513.197       95422.693
     1765569.905       95158.493     1765690.107       94913.001
#Sta/Elev= 30
     1.1 1841.89    11.4 1831.92    68.1 1803.59    79.4 1791.52   113.3 1780.15
   124.7 1764.39   147.4 1751.38   158.7  1737.9   181.3 1733.27   192.7 1715.82
   215.3 1709.29     238 1686.93   260.6 1678.61     272 1664.07   293.8 1663.49
   304.1 1652.12   324.8 1646.62   345.5    1631   400.1 1622.71   407.6 1622.58
   415.1  1622.6   531.7 1634.96   574.7 1654.29     586  1666.8   608.5 1668.58
   698.6 1695.82   733.8 1696.46   756.8 1707.44   779.8  1705.1   828.2 1717.54
#Mann= 3 , 0 , 0
       0     .08       0   400.1    .045       0   415.1     .08       0
Bank Sta=400.1,415.1
XS Rating Curve= 0 ,0
Exp/Cntr=0.3,0.1

Type RM Length L Ch R = 1 ,14078.8 ,87.9,102.7,117.4
XS GIS Cut Line= 4
     1765417.072       95677.073     1765632.843       95408.417
     1765656.112       95253.993     1765802.075       95027.646
#Sta/Elev= 30
      .4 1820.71    13.3 1810.59    30.5 1809.35    52.2  1782.3    78.2 1778.29
    95.1 1760.04   117.1 1755.38   143.1 1730.05   159.7 1729.16     182 1700.29
   207.9 1695.81   224.3 1677.58   246.9 1672.37   272.8 1655.31   288.9 1654.43
   311.7  1638.5   433.9 1624.85   441.4 1622.54   448.9 1628.29   515.2 1645.67
   527.2 1656.25   551.3 1662.72   563.3 1675.49   587.4 1683.04   611.5 1702.63
   635.6 1704.06   654.8 1729.78   671.7 1730.16   695.7 1750.15     770 1782.19
#Mann= 3 , 0 , 0
      .4     .08       0   433.9    .045       0   448.9     .08       0
Bank Sta=433.9,448.9
XS Rating Curve= 0 ,0
Exp/Cntr=0.3,0.1

Type RM Length L Ch R = 1 ,13976.1 ,186.3,180.2,174.1
XS GIS Cut Line= 4
     1765451.606       95708.652     1765653.977       95457.888
     1765834.352       95281.913     1765891.544       95053.145
#Sta/Elev= 30
     1.9 1811.51    27.9 1803.11    39.8 1789.36    92.9 1760.61   104.3 1760.61
   131.9 1736.29   183.9 1704.24   209.9 1694.23   222.9 1680.29   233.1 1680.15
   261.9 1663.01   328.8 1636.68   385.4 1631.24   406.8 1623.22   414.3 1621.98
   421.8 1621.99   457.8 1642.22   530.2 1668.03   554.9 1687.87   584.3 1696.32
   594.7 1710.87   615.5  1714.3     626 1732.89   646.8 1738.66   667.7 1755.86
   688.5  1760.7   698.9 1775.19   719.8 1779.58   730.2 1794.61     810 1823.72
#Mann= 3 , 0 , 0
     1.9     .08       0   406.8    .045       0   421.8     .08       0
Bank Sta=406.8,421.8
XS Rating Curve= 0 ,0
Exp/Cntr=0.3,0.1

Type RM Length L Ch R = 1 ,13795.9 ,118.5,119.2,120
XS GIS Cut Line= 4
     1765552.662       95788.883      1765777.16       95642.661
     1765906.943       95420.555     1766126.513       95203.001
#Sta/Elev= 30
     1.5 1811.29      42  1783.5    54.1  1783.5    66.2 1768.51   131.2 1747.78
   162.7 1726.79     187 1723.04   223.9 1696.29   247.2 1693.46   275.2 1671.78
   406.5 1621.35     414 1619.31   421.5 1621.18   462.7 1632.58   474.4 1641.99
   497.8 1643.12   514.3 1659.13   577.9 1680.72   592.2 1689.14   606.6 1707.08
   617.1 1707.08   674.1 1745.18   688.3 1747.51   707.2 1769.47     731 1775.76
   750.3 1812.78   779.1 1807.47   802.2 1822.66   822.2 1809.34   834.3 1810.99
#Mann= 3 , 0 , 0
       0      .1       0   406.5    .045       0   421.5      .1       0
Bank Sta=406.5,421.5
XS Rating Curve= 0 ,0
Exp/Cntr=0.3,0.1

Type RM Length L Ch R = 1 ,13676.7 ,108,106.7,105.5
XS GIS Cut Line= 4
     1765705.666       95836.112     1765912.909       95640.071
      1766016.53       95474.837     1766148.158       95281.597
#Sta/Elev= 30
       5 1770.47    25.8 1763.94    55.2 1743.01    74.6  1740.2    99.4 1716.54
   116.3 1714.09   158.1 1686.33     186 1677.51   199.9 1664.72   227.7 1660.74
   246.6 1650.96   301.6 1642.77   329.9 1623.36   337.4 1617.92   344.9 1618.05
   373.3 1627.28   480.3 1645.41     493 1659.65   517.4 1657.02   529.7 1676.53
   554.2 1685.97   578.6 1713.49   603.1 1715.64   615.4 1736.43   639.8  1735.7
   652.1 1751.76   664.3 1759.13   676.5 1758.53     701 1769.14   713.3 1765.62
#Mann= 3 , 0 , 0
       0      .1       0   329.9    .045       0   344.9      .1       0
Bank Sta=329.9,344.9
XS Rating Curve= 0 ,0
Exp/Cntr=0.3,0.1

Type RM Length L Ch R = 1 ,13570   ,182,183.3,184.6
XS GIS Cut Line= 4
     1765763.962       95902.225     1766005.927       95699.853
     1766120.311       95493.083     1766203.899       95237.919
#Sta/Elev= 30
     4.5 1764.82    34.2 1760.63    51.8 1746.32    83.3 1739.54   113.3 1719.63
   130.6 1718.95   162.2 1701.68   193.7 1696.49   218.8 1673.93     241 1672.67
   256.8 1658.74   341.8 1633.01   353.3 1619.59   374.6 1618.24   382.1 1617.85
   389.6 1620.65   571.3 1646.42   581.9 1665.25   603.2 1666.28   613.9 1681.16
   624.5 1688.35   635.2 1688.24   656.4 1707.51   677.7 1708.17   688.4 1727.31
   709.7 1727.25     731 1745.15   762.9 1754.21   784.2 1749.74   820.2 1753.96
#Mann= 3 , 0 , 0
       0      .1       0   374.6    .045       0   389.6      .1       0
Bank Sta=374.6,389.6
XS Rating Curve= 0 ,0
Exp/Cntr=0.3,0.1

Type RM Length L Ch R = 1 ,13386.7 ,110.8,108.6,107.2
XS GIS Cut Line= 4
     1765947.567       96056.542     1766133.509       95831.835
     1766274.289       95607.467     1766333.185       95332.395
#Sta/Elev= 30
     6.8 1841.76    22.9 1819.27    46.5 1814.71    71.7 1791.33    86.3 1790.64
   112.2 1765.23   133.9 1763.38   151.5 1742.42   177.8 1734.09   204.1 1712.27
   217.2  1709.7   243.4 1686.28   269.7 1679.02   282.8 1664.35   307.5 1654.17
   331.4 1638.26   349.9 1638.07   367.2 1626.38   391.1 1625.36   418.5 1616.41
     426  1616.4   433.5  1617.4   599.4 1653.27   754.9 1671.21   764.9 1674.05
   775.3 1682.79     796 1681.95   806.3 1690.81     827 1689.41   837.8 1693.93
#Mann= 3 , 0 , 0
       0      .1       0   418.5    .045       0   433.5     .08       0
Bank Sta=418.5,433.5
XS Rating Curve= 0 ,0
Exp/Cntr=0.3,0.1

Type RM Length L Ch R = 1 ,13278.1 ,123,126.8,129.8
XS GIS Cut Line= 4
     1766024.932       96116.171     1766226.574       95883.722
     1766344.199       95687.681     1766425.415       95432.828
#Sta/Elev= 30
     5.9 1826.21    27.7 1805.15      46 1803.02    59.4 1788.59      74 1781.14
    86.2 1781.14   104.9 1760.02   135.7 1750.39   152.2 1729.69   179.9 1724.01
   193.3 1707.47   212.9 1705.23   233.5 1687.03   259.2 1679.96   287.1 1657.67
   313.1 1651.11   324.8 1638.97   344.2 1637.72   363.9 1625.61   398.4 1619.46
   407.5 1616.39   413.4 1616.42   501.8 1626.65   525.4 1637.37   546.8 1637.44
   558.4 1643.91   579.6 1646.17   600.8 1657.07   677.2 1673.44   803.8 1685.68
#Mann= 3 , 0 , 0
     5.9      .1       0   398.4    .045       0   413.4     .08       0
Bank Sta=398.4,413.4
XS Rating Curve= 0 ,0
Exp/Cntr=0.3,0.1

Type RM Length L Ch R = 1 ,13151.2 ,287.3,292.5,297.7
XS GIS Cut Line= 4
     1766148.837       96217.091      1766276.91       95994.105
     1766497.947       95696.757     1766538.659       95443.997
#Sta/Elev= 30
     4.8 1823.66    16.5 1809.93    39.8 1806.06    51.5 1785.29    74.8 1780.34
    98.2 1760.11   133.1 1737.24   156.5 1732.42   168.1 1715.94   191.5 1712.83
   214.8 1692.14   238.1 1686.71   249.8 1677.29     287 1658.54   312.2 1651.36
   362.6 1626.91   375.2  1616.7   396.1 1616.57   403.6 1616.35   411.1 1616.81
   526.5 1623.62   543.4 1633.52   564.3 1636.31   589.5 1646.52   614.7 1648.32
   627.3 1664.82   647.9 1665.08   658.1 1679.88   699.1 1694.75   883.7  1713.8
#Mann= 3 , 0 , 0
     4.8     .08       0   396.1    .045       0   411.1     .08       0
Bank Sta=396.1,411.1
XS Rating Curve= 0 ,0
Exp/Cntr=0.3,0.1

Type RM Length L Ch R = 1 ,12858.7 ,210.6,227.7,244.8
XS GIS Cut Line= 4
     1766168.704       96240.977     1766503.057       95981.413
     1766701.029       95814.237     1766771.419       95361.102
#Sta/Elev= 30
     7.4 1821.82      33 1814.32    62.3  1785.1    95.3 1774.04   111.8 1752.65
   135.5 1748.27   199.5 1711.14   289.1 1646.77   527.3 1614.62   534.8 1614.45
   542.3 1614.83   688.4 1648.98   770.3 1687.43   790.8 1687.75     801 1706.02
   821.5 1708.81     842  1733.8   862.4 1741.27   872.7 1761.65   893.1 1761.68
   903.4 1782.82   923.8 1785.45   944.3 1805.58   964.8  1810.5     975  1824.8
   995.5  1824.8  1005.7 1841.64  1026.2  1843.6  1046.7 1860.73    1141 1891.06
#Mann= 3 , 0 , 0
       0     .08       0   527.3    .045       0   542.3      .1       0
Bank Sta=527.3,542.3
XS Rating Curve= 0 ,0
Exp/Cntr=0.3,0.1

Type RM Length L Ch R = 1 ,12631.1 ,392.6,385.1,377.7
XS GIS Cut Line= 4
     1766188.864       96294.172     1766476.661       96122.193
     1766806.614       96139.791     1767009.588       96078.406
#Sta/Elev= 30
     6.9 1839.77      54  1797.6    65.8 1797.38   101.2 1772.85     113 1752.71
   136.5 1746.84   148.3 1732.73   195.4 1710.29   207.2 1693.75     219 1693.43
   242.6 1673.09   289.7 1655.16   301.5 1639.18   470.9 1614.38   478.4 1614.34
   485.9 1614.97   539.2 1620.61   589.9 1643.17     600 1654.47   620.2 1658.04
   630.4  1672.3   671.1 1686.78   681.7 1698.64   702.8 1702.91   713.4 1717.27
   755.7 1733.15   766.2 1744.84   787.4 1746.42   797.9 1758.07   877.7  1784.6
#Mann= 3 , 0 , 0
     6.9     .08       0   470.9    .045       0   485.9     .08       0
#XS Ineff= 2 , 0
          441.75 1631.89
Permanent Ineff=
       F       F
Bank Sta=470.9,485.9
XS Rating Curve= 0 ,0
Exp/Cntr=0.3,0.1

Type RM Length L Ch R = 1 ,12246   ,312.1,317.5,322.9
XS GIS Cut Line= 4
     1766351.626       96643.846     1766573.447       96491.741
     1766899.001       96403.753     1767277.347       96210.181
#Sta/Elev= 30
     6.1 1692.42    55.1 1676.81   100.2 1675.77     141 1688.28   171.8 1672.36
   189.9 1655.67   202.3 1655.55   214.6 1645.19   251.4 1630.84   285.4 1622.41
   443.1 1608.25   450.6 1608.15   458.1 1609.53   463.5 1610.11     474  1626.4
   494.9 1632.63   505.4 1646.88   547.3 1660.54   589.2 1684.28   667.3 1711.06
   701.4 1731.67   724.1 1735.92   769.6 1768.92     815 1782.26   826.4 1795.71
   860.5 1812.58   914.2 1830.83   958.6 1832.48   980.8 1843.79  1031.2 1852.08
#Mann= 3 , 0 , 0
       0     .08       0   443.1    .045       0   458.1     .08       0
Bank Sta=443.1,458.1
XS Rating Curve= 0 ,0
Exp/Cntr=0.3,0.1

Type RM Length L Ch R = 1 ,11928.5 ,133.5,138.6,143.7
XS GIS Cut Line= 4
     1766362.058       96762.552     1766630.639       96764.502
     1767000.186       96755.703     1767369.734       96628.122
#Sta/Elev= 30
     4.7 1696.71   105.8 1669.37     116 1659.51   196.9 1636.89   267.7 1633.22
   308.2 1617.12   381.6 1606.65   389.1 1604.36   396.6 1604.37   429.6 1606.18
   439.7 1617.82   459.9 1620.51     470 1628.56   510.5 1639.31   520.6 1650.08
   591.5 1672.23   601.6 1683.33   674.4  1707.9   685.1 1723.73   738.6 1744.03
     760 1745.56   770.7 1752.85   813.8 1754.85   844.8 1764.57   856.3 1774.98
   888.4 1780.47   899.1 1776.46   968.7 1804.32  1016.8  1803.8  1029.2 1811.23
#Mann= 3 , 0 , 0
     4.7     .08       0   381.6    .045       0   396.6     .08       0
Bank Sta=381.6,396.6
XS Rating Curve= 0 ,0
Exp/Cntr=0.3,0.1

Type RM Length L Ch R = 1 ,11789.9 ,313.2,313.2,313.2
XS GIS Cut Line= 4
     1766266.291       96824.021     1766639.068       96874.526
     1766850.709       96917.816     1767091.209       96997.181
#Sta/Elev= 30
     4.6 1747.52    40.1 1742.67    50.3 1732.78    70.8 1729.53      81 1717.08
    91.2 1717.08   111.6 1703.57   121.8 1703.42     132 1693.74   203.4 1667.02
   213.7 1656.32   234.1 1652.81   244.3 1644.19   325.9 1622.13   397.6 1618.55
   483.1 1604.54   490.6    1604   498.1  1604.1   521.5    1618   531.9 1618.19
   542.2 1631.83   562.8 1636.31   573.2 1648.89   583.5 1650.43   604.5  1665.8
   666.8 1674.47     711 1691.45   763.6 1695.25   796.2 1710.38   845.5 1717.96
#Mann= 3 , 0 , 0
     4.6     .08       0   483.1    .045       0   498.1     .08       0
Bank Sta=483.1,498.1
XS Rating Curve= 0 ,0
Exp/Cntr=0.3,0.1

Type RM Length L Ch R = 1 ,11476.7 ,459.1,441.9,424.7
XS GIS Cut Line= 4
     1766123.293       97226.085     1766405.782       97124.647
     1766829.063       97216.037     1767007.608       97302.492
#Sta/Elev= 30
      .7 1843.97    11.5 1831.51    54.5 1822.52    65.1 1805.56    86.7 1800.75
    97.5 1786.76   140.5 1778.57   151.2 1760.93   172.7 1754.73   183.4 1735.11
   215.7  1710.8   226.4 1710.33   237.2 1693.48     470 1601.73   477.5 1601.56
     485 1602.16   560.3 1609.79   643.1 1635.95   653.4 1651.21   726.1 1681.32
   736.5 1694.39   752.4 1692.71   798.8 1717.96   815.2 1716.92   826.4  1732.5
   848.9 1735.96   860.1 1749.33   905.1 1760.69   916.3 1775.01   931.6 1777.01
#Mann= 3 , 0 , 0
       0      .1       0     470    .045       0     485     .08       0
Bank Sta=470,485
XS Rating Curve= 0 ,0
Exp/Cntr=0.3,0.1

Type RM Length L Ch R = 1 ,11034.7 ,286,292.7,299.4
XS GIS Cut Line= 4
     1766225.896       97692.771     1766586.645       97613.582
     1766888.895       97429.598     1767202.558        97345.22
#Sta/Elev= 30
     1.9 1794.46   144.2 1778.88   227.1 1760.19   237.4 1742.85   258.1 1737.49
   268.5 1721.34   309.9 1698.11   320.3 1676.66     479 1610.72   542.5 1601.22
     550 1600.97   557.5 1602.12   609.3 1610.75   680.3 1644.12   692.1 1661.56
   736.9 1678.02   748.1 1693.51   769.1 1700.81   779.5 1717.64   821.4 1736.95
   831.9 1751.97   852.9 1756.55   863.3 1772.32   905.2 1791.29   915.7 1805.74
   936.6 1811.14   947.1 1824.23     989 1839.46   999.5 1853.12    1048 1879.96
#Mann= 3 , 0 , 0
       0     .08       0   542.5    .045       0   557.5     .08       0
Bank Sta=542.5,557.5
XS Rating Curve= 0 ,0
Exp/Cntr=0.3,0.1

Type RM Length L Ch R = 1 ,10742.1 ,295.2,290.5,285.8
XS GIS Cut Line= 4
     1766471.679       98030.318     1766639.438        97837.95
     1767074.976       97723.566     1767312.542       97503.597
#Sta/Elev= 30
       5 1655.46    95.4 1657.64   143.3 1645.94   170.1 1645.28   297.5 1622.81
     423 1614.93   467.8 1599.49   475.3 1599.44   482.8 1603.83   558.5 1622.21
   569.4 1630.78   590.3  1635.4   600.8 1644.34     674 1658.38   694.9 1667.69
   719.1 1684.35   740.5  1690.1   755.4  1700.4   770.3 1719.06     800 1723.39
   814.9 1748.77   844.7 1754.22   856.9 1772.03   874.5    1788   904.3 1799.88
   919.1 1821.48   948.9 1825.26   967.2 1847.92   993.6 1852.63  1029.3 1872.26
#Mann= 3 , 0 , 0
       0     .08       0   467.8    .045       0   482.8     .08       0
Bank Sta=467.8,482.8
XS Rating Curve= 0 ,0
Exp/Cntr=0.3,0.1

Type RM Length L Ch R = 1 ,10451.6 ,187.3,171.1,154.8
XS GIS Cut Line= 4
     1766586.645       98308.683     1766745.023       98137.107
     1767096.973       97965.532     1767303.106       97822.437
#Sta/Elev= 30
     2.7 1776.19      39 1781.22    48.6 1780.71    63.5 1774.67   108.3 1745.11
   195.4  1681.8   233.5  1661.8     274 1632.33   285.2 1625.52   307.8 1615.24
   360.9 1600.02   389.5 1597.99     397 1597.96   404.5 1598.28   469.7 1606.11
   487.9 1610.79   555.4 1637.29     683 1692.78   708.9 1707.92   721.2 1709.34
   733.5    1721   758.1 1725.36   770.4 1738.31   782.8 1738.23   807.2 1752.46
   819.7 1749.58     832 1760.55   856.6 1763.69     869 1774.34     876 1773.15
#Mann= 3 , 0 , 0
       0     .08       0   389.5    .045       0   404.5     .08       0
Bank Sta=389.5,404.5
XS Rating Curve= 0 ,0
Exp/Cntr=0.3,0.1

Type RM Length L Ch R = 1 ,10280.5 ,268.1,268.9,269.8
XS GIS Cut Line= 4
     1766907.799       98550.649     1766925.264       98295.886
     1767040.704       98045.765     1767347.737       97868.745
#Sta/Elev= 30
     1.2 1814.51    92.4 1751.28   137.2  1722.4   163.4 1708.85   255.4 1668.71
   310.3 1635.19   332.5 1620.02   354.8 1602.36   359.9 1599.89   369.6  1598.1
   377.1 1597.92   384.6 1598.02   451.4 1601.89   467.4 1604.89   605.2 1657.54
   671.1 1687.74     698 1701.46   757.7 1734.56   768.7 1742.17   780.4  1747.7
     792  1756.7   798.2 1759.26   815.4 1760.86   827.1 1770.57   838.7 1771.83
   846.1 1778.71   858.9  1793.4   862.1 1795.25   873.8 1795.25   885.2  1804.1
#Mann= 3 , 0 , 0
     1.2     .08       0   369.6    .045       0   384.6     .08       0
Bank Sta=369.6,384.6
XS Rating Curve= 0 ,0
Exp/Cntr=0.3,0.1

Type RM Length L Ch R = 1 ,10011.6 ,677.2,692.9,708.7
XS GIS Cut Line= 4
     1767139.988       98645.164     1767160.954       98363.226
      1767302.85        98081.84     1767664.796       97991.147
#Sta/Elev= 30
     4.7 1787.42    65.5 1752.62   132.3    1717   207.5 1680.37   245.6 1663.23
   282.7 1647.21   320.9 1628.16   357.3 1610.83   368.7 1606.09     380 1601.94
   383.4 1601.08   388.7 1599.86   396.2 1598.78   417.8 1596.54   425.3 1596.17
   432.8 1597.31   436.6 1597.99   441.4 1600.09     448 1603.95   459.3 1611.19
   493.3 1628.29   527.3 1645.97   597.9 1685.08   675.6 1712.84   808.2 1762.98
   846.6 1775.97   894.6 1790.81   916.6 1798.05   941.4 1807.15     971 1819.23
#Mann= 3 , 0 , 0
       0     .08       0   417.8    .045       0   432.8     .08       0
Bank Sta=417.8,432.8
XS Rating Curve= 0 ,0
Exp/Cntr=0.3,0.1

Type RM Length L Ch R = 1 ,9318.6  ,153.3,155.7,158.2
XS GIS Cut Line= 4
     1767272.948       98942.193     1767497.316       98814.611
     1767800.873        98682.63     1768025.241       98374.674
#Sta/Elev= 30
     7.2 1693.57    28.1 1684.79    57.8 1670.46    83.3 1660.77   179.3 1636.84
   202.6 1631.88   271.7 1609.49   304.8 1602.48   359.9 1594.04     404 1593.93
   418.6 1592.33   426.1 1591.84   433.6 1594.47   438.3 1596.16   448.1 1603.76
   459.2 1611.01     551 1654.75   649.8 1704.68   661.6 1710.21   678.8 1715.24
   703.8 1719.18   741.3 1722.33   764.7 1726.54   816.2 1742.01     838 1749.59
     854 1751.83   888.7 1753.58   910.4 1752.27   941.6 1747.35   970.1 1740.83
#Mann= 3 , 0 , 0
       0     .08       0   418.6    .045       0   433.6      .1       0
Bank Sta=418.6,433.6
XS Rating Curve= 0 ,0
Exp/Cntr=0.3,0.1

Type RM Length L Ch R = 1 ,9162.9  ,392.1,381.1,370.1
XS GIS Cut Line= 5
     1767329.476       99086.418     1767562.806       98939.583
     1767755.792       98879.431      1767847.48       98747.446
     1767998.042       98560.834
#Sta/Elev= 30
     1.6 1775.75    21.8 1765.22    39.5 1754.49    93.5  1718.3     168 1669.45
   195.7 1654.15   221.5 1640.67   248.4  1627.7   283.7 1612.35   304.9 1604.55
   347.3  1595.5     379 1587.89   416.2 1585.39   423.7 1584.92   431.2 1584.93
   439.8  1586.3   447.9  1589.6   463.3 1598.06     502  1617.3   534.7 1633.34
     543 1636.78     547  1638.4   571.7 1644.55   581.7 1647.63   596.2  1653.5
   613.9 1659.62   638.5 1664.51     683 1671.29   790.9 1677.65   878.3 1681.82
#Mann= 3 , 0 , 0
       0     .08       0   416.2    .045       0   431.2      .1       0
Bank Sta=416.2,431.2
XS Rating Curve= 0 ,0
Exp/Cntr=0.3,0.1

Type RM Length L Ch R = 1 ,8781.8  ,127.4,121.1,114.7
XS GIS Cut Line= 4
     1767533.731        99344.47     1767788.662       99293.964
     1767928.152       99154.474     1768077.263       98904.353
#Sta/Elev= 30
     1.9 1670.97    16.8 1664.52    26.2 1661.93    68.4 1656.23   109.6 1654.87
   119.9 1653.23   130.2 1650.38   171.5 1636.71   181.8 1632.58   191.3 1627.78
     223 1608.48   233.3 1603.51   259.9 1593.87   268.5 1588.99   282.8 1582.32
   323.2 1571.23   332.5 1569.87     340 1569.68   347.5 1570.24   374.5 1574.18
   403.1 1577.05     446 1580.78   466.7 1581.58   478.5 1584.74   525.6 1604.38
     549 1615.22   619.8 1653.43   631.6 1659.18   655.1 1667.29   748.2 1693.99
#Mann= 3 , 0 , 0
     1.9     .08       0   332.5    .045       0   347.5     .08       0
#XS Ineff= 2 , 0
                          370.38         1586.32
Permanent Ineff=
       F       F
Bank Sta=332.5,347.5
XS Rating Curve= 0 ,0
Exp/Cntr=0.3,0.1

Type RM Length L Ch R = 1 ,8660.7  ,286.8,276,265.3
XS GIS Cut Line= 4
     1767633.696       99672.489     1767862.464       99443.722
      1768031.13       99138.375     1768168.198        98915.62
#Sta/Elev= 30
     5.5  1854.3    91.3 1787.53   125.1 1762.17   153.7 1742.36   182.3  1724.3
   196.6 1715.82     211 1707.86   261.3 1681.37   282.5  1669.5   312.4  1652.1
   351.3 1627.91   386.6 1607.55     404 1598.04   424.3 1587.59   443.8 1578.55
   455.3 1574.24   466.9 1570.52   476.3 1569.03   483.8 1568.88   491.3  1569.2
   599.4 1577.72   617.8 1578.29   625.3 1578.93   628.7 1579.47   640.1 1583.26
   719.8  1624.4   787.6 1659.94   846.4 1687.53   900.6 1715.09   933.9 1731.39
#Mann= 3 , 0 , 0
     5.5      .1       0   476.3    .045       0   491.3     .08       0
#XS Ineff= 2 , 0
                          534.11          1593.9
Permanent Ineff=
       F       F
Bank Sta=476.3,491.3
XS Rating Curve= 0 ,0
Exp/Cntr=0.3,0.1

Type RM Length L Ch R = 1 ,8384.7  ,253.5,266.7,280
XS GIS Cut Line= 4
     1767952.513       99775.065     1768197.513         99455.1
     1768207.133       99224.219     1768381.705       98975.695
#Sta/Elev= 30
     2.1 1784.67      53 1776.38    91.3 1768.65   129.5 1763.38   142.2 1760.55
   147.1 1758.02   159.6 1754.58   180.4 1743.17   244.1 1701.34   286.6 1676.63
   336.6 1651.74   349.1  1646.7   384.3 1636.35     403 1628.22   438.7  1593.9
     459 1576.47   469.1 1571.12   479.2 1569.27   512.2 1567.62   519.7  1567.3
   527.2 1568.23   550.1 1575.67   560.2 1577.52   679.9 1582.77   692.2 1584.49
   704.6 1588.29   729.3 1599.48   835.6 1654.59   863.8 1672.58   937.8 1715.26
#Mann= 3 , 0 , 0
       0      .1       0   512.2    .045       0   527.2     .08       0
Bank Sta=512.2,527.2
XS Rating Curve= 0 ,0
Exp/Cntr=0.3,0.1

Type RM Length L Ch R = 1 ,8117.9  ,222.3,249.3,275.7
XS GIS Cut Line= 4
     1767997.897       99784.586     1768365.548       99527.026
     1768526.999       99293.964     1768769.905       99183.334
#Sta/Elev= 30
     9.2 1750.66    72.4 1726.94   107.6 1712.51   132.7 1703.12     145  1699.1
   238.5 1672.83   296.6 1652.18   340.2 1639.61   354.7 1634.45   405.6 1613.67
   448.9 1589.61   478.2 1578.62   491.4 1571.31     500 1567.84   509.2 1566.01
   544.7 1566.05   621.6 1563.13   629.1 1563.08   636.6  1563.8   667.2 1569.61
   727.5 1574.44   747.1 1577.23   763.2 1582.39   801.4 1598.39   816.7 1602.39
   837.3 1605.03   847.2 1607.66   869.1 1617.83   900.7 1634.06   999.3 1686.58
#Mann= 3 , 0 , 0
     9.2     .08       0   621.6    .045       0   636.6     .08       0
#XS Ineff= 2 , 0
          534.86 1583.82
Permanent Ineff=
       F       F
Bank Sta=621.6,636.6
XS Rating Curve= 0 ,0
Exp/Cntr=0.3,0.1

Type RM Length L Ch R = 1 ,7868.6  ,357.9,362.3,366.6
XS GIS Cut Line= 4
     1767994.717       99827.243     1768349.029       99548.895
     1768719.399       99599.403     1768947.876        99474.34
#Sta/Elev= 30
      .7 1744.96    87.1 1715.17   161.2 1690.79   218.1 1675.31   276.5 1660.48
   322.3 1645.67   360.9 1635.29   381.9 1628.31   427.7 1611.36   442.2 1604.65
   450.6 1600.01   491.7 1570.58   501.9 1566.06   512.1 1564.68   563.1 1561.74
   596.5 1558.45     604 1558.44   611.5 1558.89   736.7 1560.09   746.9  1560.3
   757.1 1561.68   824.4  1584.7   852.2 1592.68   885.5 1604.32   922.8 1615.58
   944.4 1621.45     956 1623.77     979 1624.52   992.9 1626.13  1084.8 1652.03
#Mann= 3 , 0 , 0
      .7     .08       0   596.5    .045       0   611.5     .08       0
Bank Sta=596.5,611.5
XS Rating Curve= 0 ,0
Exp/Cntr=0.3,0.1

Type RM Length L Ch R = 1 ,7506.3  ,422.4,425.4,428.4
XS GIS Cut Line= 3
     1767994.548       99929.501     1768322.574       99880.786
     1768813.195      100044.327
#Sta/Elev= 30
     7.5 1716.01   123.5 1650.37   154.1 1631.23   182.6 1614.57     195 1605.39
   215.5 1585.22   225.7 1579.37   235.9 1577.66   280.5 1576.68   297.3 1573.66
   338.5 1562.81   381.1 1560.46   437.6 1552.72   445.1 1552.36   452.6 1552.73
   467.8 1554.26   477.1 1556.24   483.8 1558.82   498.4 1568.39   519.7 1585.12
   551.7 1607.74   615.7  1646.6   626.4 1650.94   647.7 1653.83   658.3 1660.42
   690.3 1683.78     765 1732.09   819.6 1770.98   828.9 1776.63   848.8 1786.63
#Mann= 3 , 0 , 0
       0      .1       0   437.6    .045       0   452.6      .1       0
Bank Sta=437.6,452.6
XS Rating Curve= 0 ,0
Exp/Cntr=0.3,0.1

Type RM Length L Ch R = 1 ,7081    ,389,382.7,376.5
XS GIS Cut Line= 4
     1767930.287      100120.247     1768173.463      100255.968
     1768451.718      100394.233      1768648.55      100515.416
#Sta/Elev= 30
    14.8 1718.06   120.8 1646.49   139.3  1633.6   209.2  1583.4   222.3 1574.86
   236.6 1566.45   238.9 1565.39   248.2 1561.67   259.8 1560.55   271.4 1560.37
   282.8 1559.37   373.2 1549.19   399.6 1545.71   407.1 1545.31   414.6  1545.7
   419.4 1545.97   429.7 1548.92   444.3 1554.93   486.1 1569.81     520 1583.12
   535.2 1589.43   555.2 1600.88   587.8 1618.57   670.9 1667.58   682.7 1673.26
   694.6 1675.74   706.5 1677.14   718.4 1681.59   730.3 1688.78   820.3 1746.06
#Mann= 3 , 0 , 0
       0     .08       0   399.6    .045       0   414.6     .08       0
Bank Sta=399.6,414.6
XS Rating Curve= 0 ,0
Exp/Cntr=0.3,0.1

Type RM Length L Ch R = 1 ,6698.2  ,393.2,383.2,373.3
XS GIS Cut Line= 4
     1767780.718      100530.161     1768062.833      100643.174
     1768300.767       100692.09      1768572.74      100745.777
#Sta/Elev= 30
      .5 1708.72    32.3 1698.85    59.5 1687.81   120.4 1652.86   150.9 1636.16
   209.2 1605.57   274.7 1572.67   285.6 1568.64   296.5 1567.41   306.8 1567.01
   317.6 1565.35     365 1552.77   379.5 1548.68   392.4  1544.2   400.2 1541.95
     403 1541.66   410.5 1540.95     418 1541.22   478.1 1549.82   486.7 1551.71
   493.1 1554.18   503.4 1560.25   544.7 1589.21   572.4 1607.54   689.1 1678.49
   699.4 1684.32   709.7 1688.11   730.3 1690.87   740.6 1695.81     824 1750.35
#Mann= 3 , 0 , 0
       0      .1       0     403    .045       0     418      .1       0
Bank Sta=403,418
XS Rating Curve= 0 ,0
Exp/Cntr=0.3,0.1

Type RM Length L Ch R = 1 ,6315    ,171,177.2,182.9
XS GIS Cut Line= 4
      1767726.58      100965.893     1768089.288         101040.
     1768337.644      100984.067     1768583.034      100896.115
#Sta/Elev= 30
     5.5 1724.45    44.8 1696.68    67.8 1681.09    82.9  1671.5     140 1638.73
     233 1586.36   291.4 1552.55   294.9  1550.6   304.3 1546.69   315.5 1544.54
   336.2 1542.81   370.2 1538.91   450.1 1532.71   480.5 1529.41     488 1529.31
   495.5 1530.03   513.4 1533.95     533 1537.01   543.4  1539.8   553.8 1543.86
   574.5 1552.82   624.8    1578   682.8  1608.5   726.3 1629.18     758 1646.86
   809.1 1674.14   819.8 1679.15   868.7 1699.13   876.6 1701.42   885.2 1702.94
#Mann= 3 , 0 , 0
       0     .08       0   480.5    .045       0   495.5     .08       0
Bank Sta=480.5,495.5
XS Rating Curve= 0 ,0
Exp/Cntr=0.3,0.1

Type RM Length L Ch R = 1 ,6137.8  ,321.6,343.7,366.3
XS GIS Cut Line= 4
     1767709.296       101001.52     1768127.768      101172.276
     1768382.699      101160.251     1768551.049      101266.071
#Sta/Elev= 30
       3  1735.1    68.5 1687.27   101.3 1667.52   122.8 1655.39   146.3 1645.01
   177.8 1633.55   210.6 1618.82   308.9 1571.88   324.8 1563.89   355.8 1545.82
   363.5 1543.38   371.3 1542.22   386.9 1538.46   396.3 1535.71   407.2 1534.06
   453.9  1531.3   595.4 1525.18   602.9    1525   610.4 1525.67     613 1525.82
   618.3 1527.25   633.2 1532.93   666.6 1544.07   707.2 1556.04   726.2 1559.01
   755.6  1562.5   823.1 1569.17     847 1572.04   882.8 1577.68     906 1582.54
#Mann= 3 , 0 , 0
       0     .08       0   595.4    .045       0   610.4     .08       0
Bank Sta=595.4,610.4
XS Rating Curve= 0 ,0
Exp/Cntr=0.3,0.1

Type RM Length L Ch R = 1 ,5794.1  ,208.5,213.4,214.2
XS GIS Cut Line= 4
      1767707.17      101032.861     1767983.467      101234.806
     1768101.313      101410.372     1768293.723       101649.75
#Sta/Elev= 30
     6.1 1726.25    14.3 1720.99    18.6 1718.88    21.5 1716.57    25.5 1714.52
    43.2 1703.18    64.9 1690.31    76.9 1685.47    86.7 1680.32    94.1 1677.78
   101.1 1673.94   111.2 1669.68   248.4 1601.22   306.7 1571.61   342.2 1554.81
   383.7 1533.27   397.3 1529.08   412.9 1527.82   433.9 1521.44   438.6 1521.08
   446.1 1520.77   453.6 1521.11   569.8 1527.24   614.4 1529.03   685.6 1530.65
   698.6 1532.54   711.6 1536.34   810.4 1571.77     832 1578.07   860.8  1585.3
#Mann= 3 , 0 , 0
       0     .08       0   438.6    .045       0   453.6     .08       0
Bank Sta=438.6,453.6
XS Rating Curve= 0 ,0
Exp/Cntr=0.3,0.1

Type RM Length L Ch R = 1 ,5580.7  ,273.9,265.7,261.6
XS GIS Cut Line= 4
     1767544.173      101205.966     1767812.175      101339.693
      1767974.44      101556.046     1768153.772      101803.857
#Sta/Elev= 30
     6.8 1665.44    40.7 1644.92    75.2 1625.77   119.8  1602.7   153.7 1586.78
     165 1582.53   176.3 1579.14     211 1570.04   278.1 1550.13   299.5 1542.51
   339.4  1524.2   351.8 1521.07   366.4 1520.46   385.5    1516     390  1515.2
   394.9  1515.1   402.4 1514.96   409.9 1515.41   486.7 1520.79   516.4 1524.27
   529.1 1526.84   541.7 1531.91   561.5 1542.86   583.2 1553.85   622.8 1575.72
     651  1590.3   714.8 1622.18   779.3 1653.51   827.7 1678.07   875.8 1701.01
#Mann= 3 , 0 , 0
     6.8     .08       0   394.9    .045       0   409.9     .08       0
#XS Ineff= 2 , 0
                          474.08         1531.31
Permanent Ineff=
       F       F
Bank Sta=394.9,409.9
XS Rating Curve= 0 ,0
Exp/Cntr=0.3,0.1

Type RM Length L Ch R = 1 ,5315    ,201.7,197.7,193.8
XS GIS Cut Line= 4
     1767478.238      101334.989     1767586.415      101466.683
     1767722.812      101624.244     1767922.703      101793.564
#Sta/Elev= 30
     1.4 1637.04    24.8 1621.96    55.6 1602.49    91.5  1580.6   127.5  1559.3
   156.2 1541.29   165.2 1536.05   176.9 1530.57   191.8 1526.29   205.2  1523.6
   213.6 1522.36   223.3 1521.23   255.9 1518.52   285.5 1515.05   306.8 1513.24
   313.7 1512.94   321.2 1512.85   328.7 1513.45   335.5  1514.3     357 1518.44
   365.8 1521.37   371.4 1524.13   391.2 1536.46   417.8 1552.31   457.4 1576.42
   500.5 1604.05     558 1639.99   593.8 1660.86   629.9 1681.07   640.8 1687.68
#Mann= 3 , 0 , 0
       0     .08       0   313.7    .045       0   328.7     .08       0
Bank Sta=313.7,328.7
XS Rating Curve= 0 ,0
Exp/Cntr=0.3,0.1

Type RM Length L Ch R = 1 ,5117.2  ,273.8,268.3,262.8
XS GIS Cut Line= 4
     1767182.691      101574.296     1767485.293      101671.278
     1767662.145      101817.619      1767913.63      101980.822
#Sta/Elev= 30
     2.4 1662.86    85.8 1625.43   109.8 1613.77   162.1 1587.04   200.5 1570.26
   237.2 1555.25   255.9 1548.64   290.3 1537.82   373.7 1514.51   388.1 1511.42
   407.7  1510.4   409.7 1510.33   422.7 1510.77   431.2 1511.63   454.5 1515.74
   467.1 1519.55   480.8 1527.23   520.2 1555.14   546.4 1572.52   618.9 1614.59
     643 1630.39   667.1 1648.13   703.3 1678.57   721.6 1692.37   736.3 1700.89
   765.5 1712.58   775.6 1717.73   811.8 1739.45   823.9 1747.25   847.1 1763.39
#Mann= 3 , 0 , 0
       0     .08       0   407.7    .045       0   422.7     .08       0
Bank Sta=407.7,422.7
XS Rating Curve= 0 ,0
Exp/Cntr=0.3,0.1

Type RM Length L Ch R = 1 ,4848.9  ,71.4,72.8,74.2
XS GIS Cut Line= 4
     1767144.302      101727.718      1767367.71      101932.313
     1767541.733      102016.973      1767819.23      102108.688
#Sta/Elev= 30
     1.8 1689.86    26.9 1675.16    49.6 1660.53   106.8 1620.93   146.7 1594.73
   180.1  1571.6   191.6 1564.32   206.6 1555.47   221.4 1547.43   236.5  1539.8
   251.5 1532.96   266.5 1527.16   282.5 1522.89   345.4  1511.6   359.7 1510.47
     406 1509.98   413.5 1509.62     421 1510.32   427.2 1512.79   436.2 1519.49
   449.6 1530.45   458.9 1536.72   527.9 1580.47     557 1599.46   594.2 1624.27
   654.5 1665.53   675.8 1679.17   701.6 1694.97     761 1730.22   788.7  1748.2
#Mann= 3 , 0 , 0
       0     .08       0     406    .045       0     421     .08       0
Bank Sta=406,421
XS Rating Curve= 0 ,0
Exp/Cntr=0.3,0.1

Type RM Length L Ch R = 1 ,4776.1  ,136.9,136.1,135.3
XS GIS Cut Line= 4
     1767092.565      101798.268     1767355.952      102000.511
     1767489.997      102075.764      1767720.46      102266.249
#Sta/Elev= 30
     1.4 1697.76    66.9 1657.46    96.6  1637.3   130.6 1612.24   163.1 1590.33
   212.9 1559.15   232.7 1548.41   258.2 1537.95   270.9 1533.97   281.8 1532.98
   296.4 1534.97   309.2 1533.01   334.5 1517.76   346.1 1511.38   349.1 1510.62
   357.7  1509.1   390.4 1510.05   406.5 1508.34     414 1507.23   421.5 1508.42
   428.9 1512.73   443.7 1524.19   451.2 1528.88   533.6 1573.75   590.2 1607.66
   650.7 1646.37   666.6 1655.03   682.4 1661.42   721.4 1673.88   784.8 1681.03
#Mann= 3 , 0 , 0
       0     .08       0   406.5    .045       0   421.5     .08       0
Bank Sta=406.5,421.5
XS Rating Curve= 0 ,0
Exp/Cntr=0.3,0.1

Type RM Length L Ch R = 1 ,4640    ,351,348.9,346.9
XS GIS Cut Line= 4
     1767075.943       101824.31     1767233.665      102082.819
     1767497.052      102226.271     1767700.134      102357.922
#Sta/Elev= 30
     6.2 1696.53    85.8 1653.93    97.7 1648.38   133.8 1633.25   165.5 1618.77
   250.3 1577.04   289.1  1558.7   302.7 1552.73     325 1539.79   340.8 1529.71
   369.8 1512.26   380.8 1506.39   384.7 1504.57   392.2 1502.84   421.9 1501.53
   429.4 1501.27   436.9  1501.4   444.4 1502.67   451.8 1505.42     502 1527.11
     538 1543.51   615.6 1577.34   652.2 1592.23   659.5 1594.64   707.5 1607.34
   738.4 1614.21   769.2 1621.75   816.7 1631.14   835.3    1637   844.7 1641.78
#Mann= 3 , 0 , 0
       0     .08       0   421.9    .045       0   436.9     .08       0
Bank Sta=421.9,436.9
XS Rating Curve= 0 ,0
Exp/Cntr=0.3,0.1

Type RM Length L Ch R = 1 ,4291.1  ,354.2,362.9,371.3
XS GIS Cut Line= 4
     1766829.479      102268.123      1767085.51      102412.052
     1767350.379       102519.72     1767567.924      102622.365
#Sta/Elev= 30
     2.9 1750.41    95.8 1688.18     119 1670.99   145.7 1650.32   200.2 1609.65
   234.9 1582.53   249.7 1571.55   264.6  1561.5     304 1536.61   364.2 1501.77
   369.5 1499.15   380.4 1495.74   394.8 1494.62   402.3 1494.42   409.8 1494.44
   424.1 1495.68   467.8 1502.15   480.7 1505.11   512.3  1517.2     577 1539.75
   584.2 1542.61   599.3 1549.31   627.1 1562.87   672.7 1584.36   677.6 1586.26
   695.5 1592.76   757.3 1613.65   794.3 1627.46   804.7 1630.76   820.2 1636.71
#Mann= 3 , 0 , 0
       0     .08       0   394.8    .045       0   409.8     .08       0
Bank Sta=394.8,409.8
XS Rating Curve= 0 ,0
Exp/Cntr=0.3,0.1

Type RM Length L Ch R = 1 ,3928.1  ,281.7,289.9,298.3
XS GIS Cut Line= 4
     1766705.915       102516.23     1766963.224      102677.791
     1767163.115      102863.572     1767357.009      103083.784
#Sta/Elev= 30
     9.6 1621.19    53.4 1600.33    65.3 1595.24     171 1558.29   208.6 1544.35
     237 1534.66   318.1 1511.25   353.2 1499.64   360.4 1497.62   374.7 1496.11
   457.8  1494.5   465.3 1494.36     470 1494.38   472.8 1494.94     482 1496.92
   489.2 1500.56     495 1504.46     525 1527.57     539 1538.81   552.8  1549.2
   589.4 1572.16   637.4 1603.46   650.9 1611.85   664.3 1619.27   696.9 1635.93
   732.7 1655.82   779.8  1680.6   795.1 1687.57     853 1712.07   870.1 1719.72
#Mann= 3 , 0 , 0
       0     .08       0   457.8    .045       0   472.8     .08       0
Bank Sta=457.8,472.8
XS Rating Curve= 0 ,0
Exp/Cntr=0.3,0.1

Type RM Length L Ch R = 1 ,3638.3  ,327.9,321.2,314.3
XS GIS Cut Line= 4
     1766613.537       102585.87     1766770.387      102790.671
     1766883.267      103023.486     1767097.586      103297.941
#Sta/Elev= 30
       4 1649.72    43.3 1628.24   114.1 1597.02   126.5 1590.95   162.7 1571.48
   209.6 1548.33   237.3 1536.95   332.2 1501.08   344.6  1497.6   354.9 1496.58
   438.2 1492.79   445.7 1492.52   453.2 1492.74   460.9 1494.16   468.3  1497.6
   479.5 1504.94   490.7 1509.37     502  1511.3   516.7  1515.1   532.1 1521.55
   557.3 1534.19   581.4 1547.18   615.4  1569.3   663.6 1594.58   679.8 1603.69
   701.4 1617.96     723 1633.78   762.2 1655.24   778.6 1661.61   864.9 1684.79
#Mann= 3 , 0 , 0
       0     .08       0   438.2    .045       0   453.2     .08       0
Bank Sta=438.2,453.2
XS Rating Curve= 0 ,0
Exp/Cntr=0.3,0.1

Type RM Length L Ch R = 1 ,3317.1  ,332.4,303.5,260.7
XS GIS Cut Line= 4
     1766429.395      102691.901      1766464.67      102927.067
     1766608.122      103082.277     1766979.685      103272.762
#Sta/Elev= 30
     4.8 1631.68      55 1592.18    91.4 1567.57   127.6 1547.73   219.6 1502.86
   229.9  1499.4   240.9 1497.35     277 1494.52   304.4 1489.04   357.3 1485.54
   364.8 1484.98   372.3 1485.79  386.69 1486.91  397.41 1489.04  403.75    1492
   413.5 1505.33   450.7 1523.98   462.1 1528.38   484.8 1534.49   535.2  1544.4
   579.5 1550.06   607.1 1554.96   628.2  1561.1   700.8 1584.89   711.7 1586.66
   719.8 1586.76   742.3 1591.04   764.9 1597.48   787.4 1605.83   866.7  1641.2
#Mann= 3 , 0 , 0
     4.8     .08       0   357.3    .045       0   372.3     .08       0
Bank Sta=357.3,372.3
XS Rating Curve= 0 ,0
Exp/Cntr=0.3,0.1
